--- G103-80-00.prj (project) ---

Proj Title=G103-80-00
Current Plan=p01
Default Exp/Contr=.3,.1
English Units
Geom File=g03
Flow File=f02
Flow File=f01
Plan File=p02
Plan File=p01
Y Axis Title=Elevation
X Axis Title(PF)=Main Channel Distance
X Axis Title(XS)=Station
BEGIN DESCRIPTION:
San Jacinto River Watershed
East Fork San Jacinto River
HCFCD unit G103-80-00
(Flood Hazard, Floodway)Model
10, 2, 1, 0.2% Event
Filename G1038000.prj
Prepared by:  FTN Associates Ltd.   DATE:  February 2003
Reviewed by:     DATE:
STATUS (Final)
The boundary condition is known water surface elevation at the downstream end, obtained from the Lake Houston model. WSEl of 45.87, 48.57, 50.01, 54.16 are used for the 10, 50, 100 and 500yr profiles respectively.
section 51110.17 is a common section for Lake houston and EF San jacincto to obtain the WSELs from the Lake Houston model as the boundary condition.
7 most upstream XS were trimmed on ROB b/c no tin data was available.  This did not cause any problem with the 2% annual chance flood extending out of the cross section limits.
The known water surface elevation of 50.90' comes from the computed floodway elevation  of Lake Houston at the common section.
END DESCRIPTION:
DSS Export Rating Curves= 0
DSS Export Rating Curve Sorted= 0
DSS Export Volume Flow Curves= 0
DXF OffsetX= 0
DXF OffsetY= 0
DXF ScaleX= 1
DXF ScaleY= 10

--- G103-80-00.p01 (plan) ---

Plan Title=Floodway
Version=Version 3.0.1  Mar 2001
Short Identifier=Floodway0607
Geom File=g03
Flow File=f02
Subcritical Flow
K Sum by GR= 0
Std Step Tol= 0.01
Critical Tol= 0.01
Num of Std Step Trials= 20
Max Error Tol= 0.3
Flow Tol Ratio= 0.001
Split Flow NTrial= 30
Split Flow Tol= 0.02
Split Flow Ratio= 0.02
Log Output Level= 0
Friction Slope Method= 1
Unsteady Friction Slope Method= 2
Parabolic Critical Depth
Global Vel Dist= 0 , 0 , 0
Global Log Level= 0
CheckData=True
Encroach Param=-1 ,0,0, 2
Encroach River=G103-80-00
Encroach Reach=EF San Jacinto
Encroach Node=118228.4
       1    3910    5873
Encroach Node=117050.2
       1    4290    6475
Encroach Node=115711.3
       1    4947    6286
Encroach Node=114421.0
       1    4653    6019
Encroach Node=113367.8
       1    4866    6459
Encroach Node=111911.9
       1    5388 7118.98
Encroach Node=110189.6
       1    3707 6140.76
Encroach Node=108173.6
       1  4527.5 5771.44
Encroach Node=107791.7
       1    4540    5800
Encroach Node=107721.3
       1    4540    5800
Encroach Node=107651.0
       1    4540    5800
Encroach Node=107249.7
       1    3843    5567
Encroach Node=106611.1
       1    3468    5402
Encroach Node=104913.0
       1    2283    4445
Encroach Node=104043.6
       1    2427    4387
Encroach Node=102963.4
       1    2489    4667
Encroach Node=102148.9
       1    2277    4052
Encroach Node=101044.2
       1    2559    3894
Encroach Node=100130.0
       1    2596    3740
Encroach Node=98845.11
       1    2560    4127
Encroach Node=97707.19
       1    2745    3956
Encroach Node=96828.22
       1    2357    3500
Encroach Node=95509.50
       1    2700    4500
Encroach Node=94407.89
       1    2545    3780
Encroach Node=92882.15
       1    1990    3137
Encroach Node=91343.42
       1    1446    2527
Encroach Node=90087.30
       1    1790    3565
Encroach Node=88594.25
       1    2204    4195
Encroach Node=87213.89
       1    1820    3773
Encroach Node=85298.22
       1    2195    4250
Encroach Node=83946.74
       1     930    2539
Encroach Node=82583.35
       1    1000    2632
Encroach Node=81851.79
       1     640    3087
Encroach Node=80668.04
       1   908.1    2805
Encroach Node=79916.10
       1     910    1972
Encroach Node=78754.21
       1     655    2080
Encroach Node=77767.82
       1  502.97    2110
Encroach Node=76556.03
       1    1060    2785
Encroach Node=75526.59
       1    1500    3205
Encroach Node=74263.07
       1    2255    4395
Encroach Node=73434.88
       1    2420    3979
Encroach Node=71410.85
       1    1205    4150
Encroach Node=70314.34
       1    1420    4501
Encroach Node=68799.84
       1    1870    4150
Encroach Node=67491.99
       1    2000    3802
Encroach Node=66268.62
       1    2435    4205
Encroach Node=65134.80
       1    3415    4514
Encroach Node=63701.51
       1    3223    4603
Encroach Node=62736.58
       1    3305    5260
Encroach Node=61490.38
       1    2812    5236
Encroach Node=60012.01
       1    3451    5471
Encroach Node=56652.75
       1 2293.09    5512
Encroach Node=53751.67
       1    1000 5201.15
Encroach Node=51110.17
       1    1622 7241.44
Encroach Reach=G103-80-00_0511
Encroach Node=118228.4
       1    3910    5873
Encroach Node=117050.2
       1    4290    6475
Encroach Node=115711.3
       1    4947    6286
Encroach Node=114421.0
       1    4653    6019
Encroach Node=113367.8
       1    4866    6459
Encroach Node=111911.9
       1    5388 7118.98
Encroach Node=110189.6
       1    3707 6140.76
Encroach Node=108173.6
       1  4527.5 5771.44
Encroach Node=107791.7
       1    4540    5800
Encroach Node=107721.3
       1    4540    5800
Encroach Node=107651.0
       1    4540    5800
Encroach Node=107249.7
       1    3843    5567
Encroach Node=106611.1
       1    3468    5402
Encroach Node=104913.0
       1    2283    4445
Encroach Node=104043.6
       1    2427    4387
Encroach Node=102963.4
       1    2489    4667
Encroach Node=102148.9
       1    2277    4052
Encroach Node=101044.2
       1    2559    3894
Encroach Node=100130.0
       1    2596    3740
Encroach Node=98845.11
       1    2560    4127
Encroach Node=97707.19
       1    2745    3956
Encroach Node=96828.22
       1    2357    3500
Encroach Node=95509.50
       1    2700    4500
Encroach Node=94407.89
       1    2545    3780
Encroach Node=92882.15
       1    1990    3137
Encroach Node=91343.42
       1    1446    2527
Encroach Node=90087.30
       1    1790    3565
Encroach Node=88594.25
       1    2204    4195
Encroach Node=87213.89
       1    1820    3773
Encroach Node=85298.22
       1    2195    4250
Encroach Node=83946.74
       1     930    2539
Encroach Node=82583.35
       1    1000    2632
Encroach Node=81851.79
       1     640    3087
Encroach Node=80668.04
       1   908.1    2805
Encroach Node=79916.10
       1     910    1972
Encroach Node=78754.21
       1     655    2080
Encroach Node=77767.82
       1  502.97    2110
Encroach Node=76556.03
       1    1060    2785
Encroach Node=75526.59
       1    1500    3205
Encroach Node=74263.07
       1    2255    4395
Encroach Node=73434.88
       1    2420    3979
Encroach Node=71410.85
       1    1205    4150
Encroach Node=70314.34
       1    1420    4501
Encroach Node=68799.84
       1    1870    4150
Encroach Node=67491.99
       1    2000    3802
Encroach Node=66268.62
       1    2435    4205
Encroach Node=65134.80
       1    3415    4514
Encroach Node=63701.51
       1    3223    4603
Encroach Node=62736.58
       1    3305    5260
Encroach Node=61490.38
       1    2812    5236
Encroach Node=60012.01
       1    3451    5471
Encroach Node=56652.75
       1 2293.09    5512
Encroach Node=53751.67
       1    1000 5201.15
Encroach Node=51110.17
       1    1622 7241.44
Computation Interval=1HOUR
Output Interval=1HOUR
Run HTab= 0
Run UNet= 0
Run PostProcess= 0
UNET Theta= 1
UNET ZTol= 0.02
UNET ZSATol= 0.1
UNET MxIter= 20
UNET MaxInSteps= 20
UNET DtIC= 0
UNET DtMin= 0
UNET MaxCRTS= 20
UNET WFStab= 2
UNET SFStab= 1
UNET WFX= 1
UNET SFX= 1
UNET Convert EG Bridges=-1
UNET Use Existing IB Tables=-1
Instantaneous Interval=1HOUR
Write IC File= 0
IC Time=0
Write Velocity= 0
Write Detailed= 0

--- G103-80-00.p02 (plan) ---

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Plan Title=FEMA Effective June 2007
Short Identifier=FEMAeff0607
Geom File=g03
Flow File=f01

--- G103-80-00.f02 (steady flow) ---

Flow Title=Floodway
Version=Version 3.0.1  Mar 2001
Number of Profiles= 2
Profile Names=1PCT_100yr, 1PCTFloodway_100yrFW
River Rch & RM=G103-80-00,G103-80-00_0511        ,118228.4
   34200   34200
River Rch & RM=G103-80-00,G103-80-00_0511        ,104043.6
   34253   34253
River Rch & RM=G103-80-00,G103-80-00_0511        ,102148.9
   34357   34357
River Rch & RM=G103-80-00,G103-80-00_0511        ,98845.11
   34431   34431
River Rch & RM=G103-80-00,G103-80-00_0511        ,96828.22
   34476   34476
River Rch & RM=G103-80-00,G103-80-00_0511        ,95509.50
   34504   34504
River Rch & RM=G103-80-00,G103-80-00_0511        ,94407.89
   34529   34529
River Rch & RM=G103-80-00,G103-80-00_0511        ,92882.15
   34570   34570
River Rch & RM=G103-80-00,G103-80-00_0511        ,91343.42
   34655   34655
River Rch & RM=G103-80-00,G103-80-00_0511        ,88594.25
   34728   34728
River Rch & RM=G103-80-00,G103-80-00_0511        ,87213.89
   34786   34786
River Rch & RM=G103-80-00,G103-80-00_0511        ,85298.22
   34877   34877
River Rch & RM=G103-80-00,G103-80-00_0511        ,81851.79
   34919   34919
River Rch & RM=G103-80-00,G103-80-00_0511        ,80668.04
   34981   34981
River Rch & RM=G103-80-00,G103-80-00_0511        ,78754.21
   35004   35004
River Rch & RM=G103-80-00,G103-80-00_0511        ,77767.82
   35097   35097
River Rch & RM=G103-80-00,G103-80-00_0511        ,74263.07
   35137   35137
River Rch & RM=G103-80-00,G103-80-00_0511        ,73434.88
   35200   35200
River Rch & RM=G103-80-00,G103-80-00_0511        ,71410.85
  108500  108500
River Rch & RM=G103-80-00,G103-80-00_0511        ,70314.34
  108584  108584
River Rch & RM=G103-80-00,G103-80-00_0511        ,68799.84
  108634  108634
River Rch & RM=G103-80-00,G103-80-00_0511        ,67491.99
  108651  108651
River Rch & RM=G103-80-00,G103-80-00_0511        ,66268.62
  108727  108727
River Rch & RM=G103-80-00,G103-80-00_0511        ,65134.80
  109075  109075
River Rch & RM=G103-80-00,G103-80-00_0511        ,60012.01
  109182  109182
River Rch & RM=G103-80-00,G103-80-00_0511        ,56652.75
  109500  109500
River Rch & RM=G103-80-00,G103-80-00_0511        ,53751.67
  121700  121700
River Rch & RM=G103-80-00,G103-80-00_0511        ,51110.17
  121724  121724
Boundary for River Rch & Prof#=G103-80-00,G103-80-00_0511        , 1
Up Type= 0
Dn Type= 1
Dn Known WS=50.01
Boundary for River Rch & Prof#=G103-80-00,G103-80-00_0511        , 2
Up Type= 0
Dn Type= 1
Dn Known WS=50.9
DSS Import GetInterval= 0
DSS Import GetPeak= 0
DSS Import FillOption= 0

--- G103-80-00.f01 (steady flow) ---

Flow Title=FEMA Effective June 2007
Version=Version 3.0.1  Mar 2001
Number of Profiles= 4
Profile Names=10PCT_10yr, 2PCT_50yr, 1PCT_100yr, 0.2PCT_500yr
River Rch & RM=G103-80-00,G103-80-00_0511        ,118228.4
   10500   24500   34200   66100
River Rch & RM=G103-80-00,G103-80-00_0511        ,104043.6
   10527   24553   34253   66127
River Rch & RM=G103-80-00,G103-80-00_0511        ,102148.9
   10578   24657   34357   66178
River Rch & RM=G103-80-00,G103-80-00_0511        ,98845.11
   10611   24731   34431   66215
River Rch & RM=G103-80-00,G103-80-00_0511        ,96828.22
   10638   24776   34476   66238
River Rch & RM=G103-80-00,G103-80-00_0511        ,95509.50
   10652   24804   34504   66252
River Rch & RM=G103-80-00,G103-80-00_0511        ,94407.89
   10665   24829   34529   66265
River Rch & RM=G103-80-00,G103-80-00_0511        ,92882.15
   10685   24870   34570   66285
River Rch & RM=G103-80-00,G103-80-00_0511        ,91343.42
   10727   24955   34655   66327
River Rch & RM=G103-80-00,G103-80-00_0511        ,88594.25
   10764   25028   34728   66364
River Rch & RM=G103-80-00,G103-80-00_0511        ,87213.89
   10793   25086   34786   66393
River Rch & RM=G103-80-00,G103-80-00_0511        ,85298.22
   10839   25177   34877   66439
River Rch & RM=G103-80-00,G103-80-00_0511        ,81851.79
   10860   25219   34919   66460
River Rch & RM=G103-80-00,G103-80-00_0511        ,80668.04
   10890   25281   34981   66490
River Rch & RM=G103-80-00,G103-80-00_0511        ,78754.21
   10902   25304   35004   66502
River Rch & RM=G103-80-00,G103-80-00_0511        ,77767.82
   10948   25397   35097   66548
River Rch & RM=G103-80-00,G103-80-00_0511        ,74263.07
   10969   25437   35137   66569
River Rch & RM=G103-80-00,G103-80-00_0511        ,73434.88
   11000   25500   35200   66600
River Rch & RM=G103-80-00,G103-80-00_0511        ,71410.85
   41300   84400  108500  182800
River Rch & RM=G103-80-00,G103-80-00_0511        ,70314.34
   41308   84467  108584  182984
River Rch & RM=G103-80-00,G103-80-00_0511        ,68799.84
   41313   84507  108634  183094
River Rch & RM=G103-80-00,G103-80-00_0511        ,67491.99
   41315   84520  108651  183131
River Rch & RM=G103-80-00,G103-80-00_0511        ,66268.62
   41323   84582  108727  183300
River Rch & RM=G103-80-00,G103-80-00_0511        ,65134.80
   41358   84860  109075  184066
River Rch & RM=G103-80-00,G103-80-00_0511        ,60012.01
   41369   84946  109182  184301
River Rch & RM=G103-80-00,G103-80-00_0511        ,56652.75
   41400   85200  109500  185000
River Rch & RM=G103-80-00,G103-80-00_0511        ,53751.67
   42700   94300  121700  211500
River Rch & RM=G103-80-00,G103-80-00_0511        ,51110.17
   42935   94300  121724  211500
Boundary for River Rch & Prof#=G103-80-00,G103-80-00_0511        , 1
Up Type= 0
Dn Type= 1
Dn Known WS=45.67
Boundary for River Rch & Prof#=G103-80-00,G103-80-00_0511        , 2
Up Type= 0
Dn Type= 1
Dn Known WS=48.57
Boundary for River Rch & Prof#=G103-80-00,G103-80-00_0511        , 3
Up Type= 0
Dn Type= 1
Dn Known WS=50.01
Boundary for River Rch & Prof#=G103-80-00,G103-80-00_0511        , 4
Up Type= 0
Dn Type= 1
Dn Known WS=54.16
DSS Import GetInterval= 0
DSS Import GetPeak= 0
DSS Import FillOption= 0

--- G103-80-00.g03 (geometry) ---

Geom Title=G103-80-00 June 2007
Version=Version 3.0.1  Mar 2001

River Reach=G103-80-00      ,G103-80-00_0511
Reach XY= 30
     3194722.432    13991284.845     3194903.193    13989767.059
     3193975.332    13989255.349     3194237.151    13987893.742
     3193285.057    13987143.777     3193845.887    13985715.405
     3192934.912    13985183.952     3193567.968     13982073.73
     3192325.671    13980973.505     3191804.923    13979551.604
       3192311.2    13978824.613     3191362.801    13976463.337
     3189420.652    13974124.522     3189268.037    13972454.355
     3185228.287    13970340.315     3186479.114     13965257.42
     3185655.669    13963577.603     3186340.231    13962983.869
     3184149.661    13961198.578     3185074.389    13959448.138
     3184327.178    13957681.955     3187261.367    13957245.023
     3188279.774    13954174.313      3191760.17    13951634.199
     3195119.346    13947279.426     3194909.334     13945616.62
     3193263.117    13942833.672     3196409.017    13934935.456
     3195672.742    13933395.973     3193088.369    13931326.274

Type RM Length L Ch R = 1 ,118228.4,623.3,1178.23,1329.76
BEGIN DESCRIPTION:
411v1
Bank Station offset =      -548
Cross section trimmed on ROB due to lack of TIN data; considered limit of study.
END DESCRIPTION:
XS GIS Cut Line= 6
     3200216.884    13990286.697     3194958.663     13990971.19
     3194811.808    13991003.226     3194540.122    13991074.235
     3193931.909    13991166.143     3192248.808     13991190.54
#Sta/Elev= 30
       0  105.95  562.57  104.01  791.35   98.91  986.47   84.87 1217.43   76.77
 1276.99   78.93 2157.61   76.82 2468.76   78.94  2781.7   75.65 3166.23   78.22
 3580.81   69.36 4618.92   70.84 4798.09   68.82 5202.35    71.2 5289.77   65.35
 5461.83   62.97 5468.05   65.06 5518.05   62.11 5535.05   49.71 5548.05   48.51
 5579.05   54.96 5630.55   57.15 5640.05   61.27 5649.05   61.11 5664.05   67.97
 6073.86   68.55 6426.85   74.95 6625.92   73.48 7052.42   83.16  8032.1   82.16
#Mann= 4 ,-1 , 0
       0     .99       0 3166.23     .12       0 5518.05     .05       0
 5640.05     .12       0
Bank Sta=5518.05,5640.05
XS Rating Curve= 0
Exp/Cntr=.3,.1

Type RM Length L Ch R = 1 ,117050.2,1466.26,1338.81,539.28
BEGIN DESCRIPTION:
411v2
Bank Station offset =      -551
Cross section trimmed on ROB due to lack of TIN data; considered limit of study.
END DESCRIPTION:
XS GIS Cut Line= 6
     3200194.669    13989975.681     3195061.883    13990320.922
     3194830.332    13990234.477     3194737.712    13990002.926
     3194334.812    13989905.445     3191112.079     13989978.03
#Sta/Elev= 30
       0  101.19  839.63   99.55 1104.31   81.31 1446.73   75.67 1606.37   78.81
 1810.78    75.2 1977.74   80.38 2424.81   74.55 3605.66   82.89 3791.61   79.88
 3947.47   68.69 5466.31   67.27 5489.31   60.34 5491.31   54.59 5501.31   51.89
 5551.31   49.77 5569.31   54.64 5586.31   66.89 5953.84   63.73 6035.36   68.42
 6188.16   66.66 6233.18   61.99 6319.22   67.94 6578.26   63.33 6946.68   83.41
 7749.34   84.09 7968.38   79.71 8493.86   84.59 9137.14   78.25 9280.65   81.63
#Mann= 4 ,-1 , 0
       0     .99       0 3605.66     .12       0 5466.31     .05       0
 5586.31     .12       0
#Block Obstruct= 2 , 0
       0                    6960       0      83
Bank Sta=5466.31,5586.31
XS Rating Curve= 0
Exp/Cntr=.3,.1

Type RM Length L Ch R = 1 ,115711.3,772.98,1290.35,1116.57
BEGIN DESCRIPTION:
411v3
Bank Station offset =      -623
Cross section trimmed on ROB due to lack of TIN data; considered limit of study.
END DESCRIPTION:
XS GIS Cut Line= 6
      3199689.53    13988033.893     3194334.812    13989060.647
     3194265.348    13989085.984     3194204.843    13989411.563
     3194061.878     13989424.56     3190731.951     13989576.91
#Sta/Elev= 30
       0   93.49  551.38  104.62 1333.28   76.44 2277.16   79.38 2714.64   70.28
    3343   74.33 3524.95   70.48 3852.89   74.76 4226.36   70.01 4406.94      74
 4640.18   66.79  5298.7   67.05 5380.34   59.71 5511.91   66.19 5591.26   64.03
 5623.26   49.08 5750.26   62.38  6066.2   55.89 6159.18    64.9 6501.44   66.11
 6709.79   82.36 7787.42   78.73 8403.39    81.7 8699.37   77.86 8835.76   80.48
 8929.11   79.15 8977.05   74.24 9094.48   77.89 9153.77   70.27 9334.33   79.25
#Mann= 4 ,-1 , 0
       0     .99       0 2277.16     .12       0 5591.26     .05       0
 5750.26     .12       0
#Block Obstruct= 2 , 0
       0                    6750       0    82.5
Bank Sta=5591.26,5750.26
XS Rating Curve= 0
Exp/Cntr=.3,.1

Type RM Length L Ch R = 1 ,114421.0,1061.25,1053.18,681.34
BEGIN DESCRIPTION:
411v4
Bank Station offset =      -570
Cross section trimmed on ROB due to lack of TIN data; considered limit of study.
END DESCRIPTION:
XS GIS Cut Line= 6
      3199442.59    13987176.098     3194451.784    13988293.831
      3194123.33    13988304.886     3193970.899    13988319.825
     3193853.927    13988345.818     3189899.569    13988841.302
#Sta/Elev= 30
       0   85.86 1110.88   73.49 1576.97   78.85 1766.88   73.73 2863.01   76.89
 3185.82   67.15 3366.18   72.29  3929.7   73.13 4158.81   66.79 4843.77   65.11
 4904.78   60.51 5349.83    65.6 5416.89   59.81 5481.26    65.5 5499.26   62.89
 5518.26   51.09 5570.26   48.53 5583.26   52.79 5588.76   60.47 5606.26   64.48
 6191.11   62.58  6389.1   81.95 6536.64   83.05  7154.3   76.46 7236.89   83.06
 7650.34   76.52 7849.65   79.11 8178.36   70.67 8953.69   95.41 9701.34   91.61
#Mann= 4 ,-1 , 0
       0     .99       0 2863.01     .12       0 5481.26     .05       0
 5606.26     .12       0
#Block Obstruct= 2 , 0
       0                    6540       0      84
Bank Sta=5481.26,5606.26
XS Rating Curve= 0
Exp/Cntr=.3,.1

Type RM Length L Ch R = 1 ,113367.8,491.19,1455.93,1197.78
BEGIN DESCRIPTION:
411v5
Bank Station offset =     -1071
Cross section trimmed on ROB due to lack of TIN data; considered limit of study.
END DESCRIPTION:
XS GIS Cut Line= 6
     3199780.509    13986136.347     3194165.853    13987280.074
     3193965.876    13987409.555     3193567.608    13987693.591
     3193419.415    13987789.299     3189331.205    13988272.938
#Sta/Elev= 30
       0  100.46  869.22   74.31 3219.18   77.02 3457.29   72.03 4441.73   78.71
 4648.39   64.98 5438.57   67.04 5785.98   59.18 6031.17   62.35 6071.17   50.16
 6131.17   52.01 6146.17   64.17 6237.51   57.44 6299.98   64.76  6363.2   60.47
 6505.98   68.72 6590.03   59.81 6668.44   69.67 6694.75   80.09 6936.35   84.72
 7298.28   80.32 7399.96   70.19 7473.03   80.47 8053.04   78.71  8185.4      67
 8263.71   77.52  9394.6   94.95 9865.35   95.8810463.03   86.7210750.75   94.68
#Mann= 4 ,-1 , 0
       0     .99       0 4441.73     .12       0 6031.17     .05       0
 6146.17     .12       0
#Block Obstruct= 2 , 0
       0                    6940       0      85
Bank Sta=6031.17,6146.17
XS Rating Curve= 0
Exp/Cntr=.3,.1

Type RM Length L Ch R = 1 ,111911.9,1392.15,1722.28,787.2
BEGIN DESCRIPTION:
411v6
Bank Station offset =     -1640
Cross section trimmed on ROB due to lack of TIN data; considered limit of study.
END DESCRIPTION:
XS GIS Cut Line= 6
     3199988.459    13985733.444     3193737.412    13986863.095
     3193552.171    13986838.396     3193558.346    13986631.544
     3193139.099    13986617.232     3188156.585    13987098.318
#Sta/Elev= 30
       0  102.05  316.89  100.96  779.82    82.5 1289.03   73.67 3530.96   77.61
 3896.79   72.43 4115.08   80.75 4425.39   71.77 4654.63   75.62    5246   63.63
 6586.45   56.83 6640.45   46.84 6677.45   56.12 6681.45   65.16 7004.31    58.8
 7221.89   70.65 7462.09   73.13 7538.49   57.57 7665.57   69.74 7746.51   71.25
 7798.28   59.62 7832.08    66.1 7953.18   60.02 8029.82   61.81 8130.71   77.62
    8513   82.7810412.46   95.0910850.18   79.6711456.31   95.2612174.59   94.95
#Mann= 4 ,-1 , 0
       0     .99       0 4654.63     .12       0 6586.45     .05       0
 6681.45     .12       0
#Block Obstruct= 2 , 0
       0                   10410       0    95.3
Bank Sta=6586.45,6681.45
XS Rating Curve= 0
Exp/Cntr=.3,.1

Type RM Length L Ch R = 1 ,110189.6,1337.33,2016.01,1634.35
BEGIN DESCRIPTION:
411v7
Bank Station offset =        10
Cross section trimmed on ROB due to lack of TIN data; considered limit of study.
block is beyond flow area
END DESCRIPTION:
XS GIS Cut Line= 6
     3198558.801    13984485.742     3193892.918    13985421.518
     3193269.067    13985928.397     3191019.081     13986239.11
     3188177.573    13986441.768     3187474.548    13986416.281
#Sta/Elev= 30
       0   82.83  491.62   88.37  627.88    76.3  725.63   72.89 3052.38   74.63
 3529.55    65.4 4248.38   67.11 4908.25   62.63 4946.55   58.85 4954.55   54.14
 4965.55   55.95 4989.55   44.59 5021.55   46.91 5043.55   61.93 5085.55   67.71
 5110.55   60.47 5185.21   62.42 5261.21   55.39  5359.7   53.59  5514.3    60.4
 5671.09   57.82  6040.9   64.37 6151.12   56.58 6319.76   69.58 7072.67    70.5
 7384.75   84.42 8624.27    82.4 8935.26   77.54 9884.42   94.8311388.89   93.15
#Mann= 4 ,-1 , 0
       0     .99       0 3052.38     .12       0 4965.55     .05       0
 5043.55     .12       0
#Block Obstruct= 2 , 0
       0                    7375       0    84.5
Bank Sta=4965.55,5043.55
XS Rating Curve= 0
Exp/Cntr=.3,.1

Type RM Length L Ch R = 1 ,108173.6,329.31,381.86,367.16
BEGIN DESCRIPTION:
411v8  XS 4/4
Bank Station offset =       441
END DESCRIPTION:
XS GIS Cut Line= 6
      3197895.96    13983991.861     3196462.585    13984590.809
     3193644.792    13984590.809     3191664.492    13985023.436
     3188080.973    13985605.024     3187020.903    13985599.236
#Sta/Elev= 30
       0   90.24  488.05   73.42 2264.11   74.83 2881.11   70.57 3030.97   76.26
 3212.41   69.34 3369.73   72.73 4468.57   70.65 4486.01   56.58  4527.5   55.11
 4558.99   45.42 4621.19   52.24 4646.71   60.65 4666.51   60.29 4742.31   54.74
 4884.71   56.33 4899.77   52.96 5034.39   57.17 5382.02   55.93 5731.99   63.66
 6525.54   68.28 6740.45   74.51 6918.05   72.85 7176.48   81.14 9054.05   97.63
10283.63    96.110472.07   93.3810530.47   88.6810584.16    92.611096.81   97.56
#Mann= 4 ,-1 , 0
       0     .99       0 3369.73     .12       0  4527.5     .05       0
 4666.51     .12       0
Bank Sta=4527.5,4646.71
XS Rating Curve= 0
Exp/Cntr=.5,.3

Type RM Length L Ch R = 1 ,107791.7,192.02,140.74,153.52
BEGIN DESCRIPTION:
411s1u:  XS 3/4
Bank Station offset =       241
END DESCRIPTION:
XS GIS Cut Line= 6
     3197763.084    13983933.567     3196210.875    13984562.841
     3195043.223    13984541.865     3192694.454    13984290.752
     3187974.824    13985147.054     3186976.472    13985154.927
#Sta/Elev= 30
       0   83.35  337.07   75.85 1047.73   70.28 2314.39   74.25 3058.17   69.46
 4007.59   71.25 4269.41   67.95 4320.99   71.41 4382.37   67.04 4523.82   67.84
 4565.65    63.2 4676.24   56.55 4681.36    53.7 4683.06    56.9 4697.05    45.2
 4759.03    43.7 4767.54   55.41 4812.42    54.6  4839.9   62.32 5116.28   63.74
 5352.06    58.3 5772.24   61.43 6394.59   71.96 6775.32   72.06 7759.14   83.02
 8156.23   91.31 9581.39   96.14 10340.3   88.6110382.44   92.1111002.93   98.45
#Mann= 3 ,-1 , 0
       0     .12       0 4565.65     .05       0  4839.9     .12       0
#XS Ineff= 2 , 0
       0    4545      73    4860       0      63
Permanent Ineff=
       F       F
Bank Sta=4565.65,4839.9
XS Rating Curve= 0
Exp/Cntr=.5,.3

Type RM Length L Ch R = 3 ,107721.3,,,
BEGIN DESCRIPTION:
FM 1485 (Huffman-Cleveland Road) 411s1
END DESCRIPTION:
Bridge Culvert--1,0,-1,-1, 0
Deck Dist Width WeirC Skew NumUp NumDn MinLoCord MaxHiCord MaxSubmerge Is_Ogee
47,46,2.6,0, 24, 26, , , .95, 0, 0,0,,
     425    2750    3600  4107.5 4210.25 4286.58 4349.85 4392.99 4418.39 4458.18
 4527.03    4549 4698.72    4851 4871.37 4921.44 4971.53 5046.68 5096.61 5198.17
    5635    6350    6900    7300
    74.5    74.2      73   74.48   75.21   75.85   76.28   76.85   76.99   77.54
   78.21   78.02   78.41   78.02   78.27    77.5   76.23   74.57    72.8   68.51
      63    71.4      74      80
                                                                                
           74.22   74.61   74.22
                                
     580    2776    3626  4126.5 4229.25 4305.58 4368.85 4411.99 4437.39 4477.18
 4546.03    4568 4717.72    4870 4890.37 4940.44 4990.53 5065.68 5115.61 5217.17
    5664    6297    6850    7380    8120    8760
    74.5    74.4      73   74.48   75.21   75.85   76.28   76.85   76.99   77.54
   78.21   78.02   78.41   78.02   78.27    77.5   76.23   74.57    72.8   68.51
      63    70.6      74      80      88      91
                                                                                
           74.22   74.61   74.22
                                                
Pier Skew, UpSta & Num, DnSta & Num=  ,4599, 3 ,4618, 3 , 2 , 2 , 0 ,0,
    1.35       2       2
   72.22   72.22      75
    1.35       2       2
   72.22   72.22      75
Pier Skew, UpSta & Num, DnSta & Num=  ,4639, 3 ,4658, 3 , 2 , 2 , 0 ,0,
    1.35       2       2
   72.22   72.22      75
    1.35       2       2
   72.22   72.22      75
Pier Skew, UpSta & Num, DnSta & Num=  ,4679, 3 ,4698, 3 , 2 , 2 , 0 ,0,
    1.35       2       2
   72.22   72.22      75
    1.35       2       2
   72.22   72.22      75
Pier Skew, UpSta & Num, DnSta & Num=  ,4719, 3 ,4738, 3 , 2 , 2 , 0 ,0,
    1.35       2       2
   72.22   72.22      75
    1.35       2       2
   72.22   72.22      75
Pier Skew, UpSta & Num, DnSta & Num=  ,4759, 3 ,4778, 3 , 2 , 2 , 0 ,0,
    1.35       2       2
   72.22   72.22      75
    1.35       2       2
   72.22   72.22      75
Pier Skew, UpSta & Num, DnSta & Num=  ,4799, 3 ,4818, 3 , 2 , 2 , 0 ,0,
    1.35       2       2
   72.22   72.22      75
    1.35       2       2
   72.22   72.22      75
Abutment Skew #Up #Dn= , 4 , 4
    4549    4559    4559  4596.5
   74.22   74.22   72.22   59.87
    4568    4578    4578  4615.5
   74.22   74.22   72.22   59.87
Abutment Skew #Up #Dn= , 4 , 4
  4801.5    4839    4839    4851
    54.6   72.22   74.22   74.22
  4820.5    4858    4858    4870
    54.6   72.22   74.22   74.22
BR Coef= 1 , 1 , 1 ,1.25, 0 ,,,.8,-1,2,0,
WSPro=,,,, 1 ,,,, 0 ,,,, 0 ,,,,-1 ,-1 ,-1 , 0 , 0 , 0 , 0 , 0
BC Design=,, 0 ,, 0 ,,,,,,

Type RM Length L Ch R = 1 ,107651.0,427.51,401.3,481.55
BEGIN DESCRIPTION:
Copy of 411s1u:  XS 2/4
Bank Station offset =       222
END DESCRIPTION:
XS GIS Cut Line= 6
     3197700.156     13983507.06     3196882.101    13984108.366
     3196078.029    13984388.043     3193779.103    13984272.358
     3192226.566    13984070.316     3186865.395    13984621.756
#Sta/Elev= 30
       0   90.55     429   83.44  786.95   70.44 1627.58   72.21  1846.6   67.44
 2224.07   72.05  3442.7   70.08 3557.29   73.27 4586.63   67.83 4601.69   66.79
 4607.16   59.87 4700.48    53.7 4702.18    56.9 4716.17    45.2 4778.15    43.7
 4786.66   55.41 4831.54    54.6 4839.76   59.58 4873.46   64.19    5055    65.7
 5415.61   58.41 5920.39   62.09 5970.73   66.61 6231.69   71.26 7101.94   71.87
 8803.44   92.07 9673.81   87.97 9799.46   82.43 9916.72   88.2311126.46  100.42
#Mann= 3 ,-1 , 0
       0     .12       0 4586.63     .05       0 4873.46     .12       0
#XS Ineff= 2 , 0
       0    4560      73    4915       0      67
Permanent Ineff=
       F       F
Bank Sta=4586.63,4873.46
XS Rating Curve= 0
Exp/Cntr=.5,.3

Type RM Length L Ch R = 1 ,107249.7,809.43,638.61,474.8
BEGIN DESCRIPTION:
Copy of 411s1u:  XS 1/4
Bank Station offset =       504
END DESCRIPTION:
XS GIS Cut Line= 6
     3197745.517    13983255.597     3196628.966    13983510.808
     3193779.103    13983872.358     3192226.566    13983670.316
      3191461.93    13983810.759     3186820.964    13984332.955
#Sta/Elev= 30
       0   90.71  671.54   87.05 1073.22   74.82 2168.66   76.81 2691.12   66.22
 2758.63   70.89 3138.65   72.99 3509.86   63.78 4191.01   66.81 4313.71   54.51
 4321.19   54.62 4324.74   59.87 4412.94   56.55 4419.76    56.9 4433.75    45.2
 4495.73    43.7 4503.73   55.09 4511.72    55.5 4527.55   55.16 4995.41    55.2
 5178.15    62.9 5770.51    60.1  5990.8   68.77 6476.02   68.33 6757.73   74.81
  8514.2   86.56 9199.26   80.48 9382.21      8710255.61   91.4211032.36  101.69
#Mann= 5 ,-1 , 0
       0     .99       0 3138.65     .12       0 4412.94     .05       0
 4527.55     .12       0 6757.73     .99       0
Bank Sta=4412.94,4511.72
XS Rating Curve= 0
Exp/Cntr=.3,.1

Type RM Length L Ch R = 1 ,106611.1,1364.17,1698.08,1222.21
BEGIN DESCRIPTION:
411v9
Bank Station offset =       868
END DESCRIPTION:
XS GIS Cut Line= 6
     3197364.544    13982954.697     3194066.216    13983035.962
     3193378.325    13983085.589     3193312.376    13983146.591
     3193134.315    13983323.004     3186754.317    13983288.828
#Sta/Elev= 30
       0   87.07  608.81   87.21 1161.64   73.61 2252.16   76.43 2750.16   72.95
 2838.28   70.36 2906.64   61.02 3011.67   70.59  3272.5   63.71 3977.09   66.07
 4020.41   65.08 4049.68   58.33 4051.77   65.45 4101.77   65.15 4131.77   44.77
 4199.77   45.87 4213.27   53.57 4248.27   57.67 4423.19   53.37 4929.94    63.3
 5392.92    58.8 5997.79   71.48 7445.07   82.39 8124.24   80.28 8270.08   78.21
 8323.27   72.61 8435.09   81.59 9041.39    90.8 9515.25   89.1410709.59   98.31
#Mann= 5 ,-1 , 0
       0     .99       0 2252.16     .12       0 4101.77     .05       0
 4248.27     .12       0 7445.07     .99       0
Bank Sta=4101.77,4248.27
XS Rating Curve= 0
Exp/Cntr=.3,.1

Type RM Length L Ch R = 1 ,104913.0,165.85,869.44,556.74
BEGIN DESCRIPTION:
411v10
Bank Station offset =      2217
END DESCRIPTION:
XS GIS Cut Line= 6
     3195746.359     13981249.48     3193885.441    13981674.833
     3193247.412    13981855.608     3193170.204    13981886.136
     3193233.064     13982148.51     3186554.378    13982311.348
#Sta/Elev= 30
       0    81.9  268.36   83.55  519.27   72.61 1697.34   70.38 1752.35   67.89
 1809.45   55.99 1969.88    67.8 2111.37   70.01 2357.56   68.42 2504.85   55.28
 2729.51   57.18 2750.51   46.81 2783.01   44.11 2846.01   54.11 3581.31   61.67
 3684.77   56.38 3921.96   57.04 4276.11   67.24 5034.92   66.68 5350.26   77.29
 6335.98   80.48 6580.92   75.93 6690.91   67.17 6745.68   74.85 7000.75   79.69
 8032.29   80.94 8524.85   92.45 8833.26   87.82 8951.33   79.87 9610.94   89.58
#Mann= 6 ,-1 , 0
       0     .12       0 1697.34     .99       0 2111.37     .12       0
 2729.51     .05       0 2846.01     .12       0 6335.98     .99       0
Bank Sta=2729.51,2846.01
XS Rating Curve= 0
Exp/Cntr=.3,.1

Type RM Length L Ch R = 1 ,104043.6,1019.47,1080.17,414.8
BEGIN DESCRIPTION:
411v11
Bank Station offset =      2151
END DESCRIPTION:
XS GIS Cut Line= 6
     3195778.261    13980983.635      3193353.75    13981653.565
     3192883.232    13981618.296     3190184.873    13981653.565
     3189195.927    13981759.904     3186487.584    13981885.986
#Sta/Elev= 30
       0   84.17  267.56   84.53  651.65   73.02 1926.11   69.92 2005.19    52.6
 2091.97   62.87 2271.18   68.89 2462.93   62.74 2505.33   56.04 2827.58   56.71
 2848.58   42.81 2945.58   50.51 2955.58   56.11 2957.58   56.51 3270.52   51.93
 3501.38   63.59 4297.03   63.25 4592.36   68.84 5209.81   65.34  5622.3   77.19
 6189.05   73.35 6368.03   66.06 6488.72   73.37 7255.45   78.77 7517.31   70.86
  7856.1   80.74  8027.3   75.06 8210.94   82.82 8583.99   81.52 9393.96   96.69
#Mann= 6 ,-1 , 0
       0     .12       0 1926.11     .99       0 2271.18     .12       0
 2827.58     .05       0 2957.58     .12       0  5622.3     .99       0
Bank Sta=2827.58,2955.58
XS Rating Curve= 0
Exp/Cntr=.3,.1

Type RM Length L Ch R = 1 ,102963.4,382.26,814.52,1011.57
BEGIN DESCRIPTION:
411v12
Bank Station offset =      1749
END DESCRIPTION:
XS GIS Cut Line= 6
     3195406.077    13980632.719     3194289.526    13980611.451
     3192513.679    13980781.592     3192439.242     13981249.48
     3189280.998    13981153.776     3186453.524    13981238.838
#Sta/Elev= 30
       0    79.5  327.08   74.39 1934.46   73.14 2513.93   51.77 2706.06   53.53
 2756.08   50.38 2902.36   56.65  3000.1   49.78  3116.7   51.52 3126.38   56.88
 3167.34   53.46 3195.86   43.41 3250.54   43.09 3279.92   50.61 3286.03   58.63
  3378.8   56.66 3404.57   60.92 3587.84   65.07 3778.93   60.59 3997.52   65.22
 5208.28   63.67 5778.23   71.85 6120.52   70.09  6354.4   62.17 6488.84      70
 6827.66   75.77 7664.68   79.83 8376.12    92.9 8821.87   92.38 9370.83  101.55
#Mann= 5 ,-1 , 0
       0     .12       0 3167.34     .05       0 3279.92     .12       0
 6120.52     .99       0 6488.84     .12       0
Bank Sta=3167.34,3286.03
XS Rating Curve= 0
Exp/Cntr=.3,.1

Type RM Length L Ch R = 1 ,102148.9,923.16,1104.62,928.19
BEGIN DESCRIPTION:
411v13
Bank Station offset =      2370
Extended XS on LOB
END DESCRIPTION:
XS GIS Cut Line= 6
 3195863.525721913980324.3338356      3192355.79    13980410.267
     3192149.575    13980329.133     3191843.748    13980303.071
     3189206.561    13980292.437     3186443.301    13980467.465
#Sta/Elev= 30
   -1000      84    -630      76  182.36   72.14 1859.14   72.97  2230.2   57.88
 2285.56   51.62 2440.64   55.55 2567.01    51.1 2630.01      40 2656.01    40.9
 2677.51    56.4 2736.01    57.2 3002.42   52.42 3092.56   55.22 3166.81   51.45
  3257.6   55.63  3400.1    53.9 3617.67   66.68 3853.24   67.57 4445.58   65.85
 4519.61   61.23 4648.49   63.81 4772.91   58.08 4876.97   68.07 4961.35   69.45
 6603.61   75.53 6964.14   80.97 7231.15   90.21 7825.63   87.33 8444.11   99.91
#Mann= 3 ,-1 , 0
   -1000     .12       0 2567.01     .05       0 2736.01     .12       0
Bank Sta=2567.01,2677.51
XS Rating Curve= 0
Exp/Cntr=.3,.1

Type RM Length L Ch R = 1 ,101044.2,646.03,914.27,257.19
BEGIN DESCRIPTION:
411v14
Bank Station offset =      1835
END DESCRIPTION:
XS GIS Cut Line= 6
     3194948.823    13979303.492      3194300.16    13979335.393
     3192024.523     13979633.14     3191705.509    13979388.562
     3190089.168    13979601.239     3188068.743     13979771.38
#Sta/Elev= 30
       0   78.31  569.68   67.31  691.31   73.47  776.12   64.13  855.38   71.77
 1175.04   71.62 1275.66   60.32 1321.01   68.13  1453.7   70.75 1572.39   57.89
 1676.41   68.22 1776.09   59.68 1848.81   72.49 2544.45   59.97  2864.4   63.66
 2939.43   48.03    2975   47.86 3002.69   55.99 3103.39   55.21 3138.39   41.81
 3165.39   41.31 3194.39   45.31 3212.39   60.91 3273.39   57.11 3456.15    63.6
 4089.76    61.2 4605.72    69.9 5117.09   65.88 5344.03   71.95 7021.25   75.19
#Mann= 6 ,-1 , 0
       0     .99       0 1848.81     .12       0 3103.39     .05       0
 3212.39     .12       0 4605.72     .99       0 5344.03     .12       0
Bank Sta=3103.39,3212.39
XS Rating Curve= 0
Exp/Cntr=.3,.1

Type RM Length L Ch R = 1 ,100130.0,1169.69,1284.92,1149.31
BEGIN DESCRIPTION:
411v15
Bank Station offset =      2325
LOB block due to laterial streams.  Flow will not be conveyed downstream.
END DESCRIPTION:
XS GIS Cut Line= 6
     3194927.555    13978622.927      3193938.61    13978676.096
     3193417.553     13978824.97     3192399.738    13978916.055
     3189727.618    13979473.633     3188068.743    13979484.267
#Sta/Elev= 30
       0   81.86  562.25    73.9  868.93   82.03 1285.77   71.68 2367.84   71.78
 2412.86   65.25 2518.79   59.64 2598.42   60.14 2618.42    48.5 2638.42    42.6
 2675.42    41.2 2707.42    41.9 2726.42    50.3 2753.42    52.9 2827.45   58.27
 2873.72   49.38 2904.56   53.18 2935.41   50.86 2966.26   56.92 3115.77   57.19
 3227.96   62.05 4022.75    60.4 4513.28   69.43 4681.46   66.34 4875.65   69.47
 5034.49   65.46 5146.31   70.72 5912.53   69.41  6198.2   77.26 6947.63   76.67
#Mann= 3 ,-1 , 0
       0     .12       0 2598.42     .05       0 2753.42     .12       0
Bank Sta=2598.42,2726.42
XS Rating Curve= 0
Exp/Cntr=.3,.1

Type RM Length L Ch R = 1 ,98845.11,1117.14,1137.92,1122.36
BEGIN DESCRIPTION:
411v16
Bank Station offset =      2152
END DESCRIPTION:
XS GIS Cut Line= 6
     3194470.301    13977602.081     3193417.553    13977644.616
     3191950.086    13977846.659     3189132.125    13978452.786
     3188515.363    13978527.223 3187321.020294813978574.9976067
#Sta/Elev= 30
       0   81.36  361.06   81.83   960.4   88.16 1065.58   85.82 1273.61   74.68
 1457.73   70.23 2197.38   67.87 2338.03   60.71    2364   56.51 2433.78   60.62
 2455.44    64.5 2651.19    57.5 2707.64   51.27 2780.23   43.52 2847.73   40.42
 2867.23   40.42 2886.23   52.12  2966.4   53.37 3006.62   57.53  3069.5   49.57
 3114.99   50.69 3153.64   60.43 3725.81   59.54 3954.62   63.84 4455.57   61.64
 4695.42   66.79 5131.95    62.2 5622.15   71.82 6131.13   68.39    7235      74
#Mann= 3 ,-1 , 0
       0     .12       0 2780.23     .05       0 2847.73     .12       0
Bank Sta=2707.64,2886.23
XS Rating Curve= 0
Exp/Cntr=.3,.1

Type RM Length L Ch R = 1 ,97707.19,903.9,878.97,760.13
BEGIN DESCRIPTION:
411v17
Bank Station offset =      2101
END DESCRIPTION:
XS GIS Cut Line= 6
     3194353.329    13976666.305     3192407.341    13976698.206
     3191301.608    13976846.157     3189483.041    13977251.165
     3188653.603    13977314.968 3187011.561935213977971.7782493
#Sta/Elev= 30
       0   80.13   84.48   78.31  319.04   78.87  806.36    89.1 1265.11   87.74
 1739.77   71.63 1889.81   68.72 2238.72   69.54 2506.25   62.99 2600.48   66.92
  2698.5   59.23 2795.71   57.43 2825.71   44.53 2875.71   44.53 2898.71   35.83
 2927.71   39.43 2946.21   49.93 2955.71   58.43 3138.76   60.86 3377.66   56.92
 3451.78   58.52 3666.35   57.32 3757.18   62.09 3976.79   59.37  4265.9   60.67
 4602.53   66.43 4995.15   69.75 5986.53   67.51    7256      70    7526      74
#Mann= 3 ,-1 , 0
       0     .12       0 2795.71     .05       0 2955.71     .12       0
Bank Sta=2795.71,2955.71
XS Rating Curve= 0
Exp/Cntr=.3,.1

Type RM Length L Ch R = 1 ,96828.22,1507.54,1318.72,1097.41
BEGIN DESCRIPTION:
411v18
Bank Station offset =      2297
ROB flow will be conveyed for 500yr flood
END DESCRIPTION:
XS GIS Cut Line= 6
     3193747.202    13975847.501     3192513.679    13975911.304
     3191171.213    13975919.609     3191049.103    13976177.186
     3188653.603    13976528.065 3186562.063069113977693.9193696
#Sta/Elev= 30
       0   73.83  311.12   68.47 1343.01   71.33 1572.48   63.03 1675.72   66.29
  1798.2   67.42  2118.5   59.66 2334.95   62.11 2418.08   58.84 2470.07   52.61
 2543.98   57.58 2648.22   49.75 2658.22   46.05 2661.22   37.85 2703.22   36.55
 2740.22   37.55 2745.72   47.05 2763.22   56.35 2799.72   53.65 2854.03   59.53
 3175.07   58.81 3259.44   57.13 3336.87   50.05 3495.28   50.36 3547.03   53.34
  3602.5   65.51 3876.04   71.62  5670.7   67.54    7200      70    7680      74
#Mann= 4 ,-1 , 0
       0     .99       0 1675.72     .12       0 2648.22     .05       0
 2763.22     .12       0
Bank Sta=2648.22,2763.22
XS Rating Curve= 0
Exp/Cntr=.3,.1

Type RM Length L Ch R = 1 ,95509.50,1428.55,1101.61,867.19
BEGIN DESCRIPTION:
411v19
Bank Station offset =      1326
ROB flow will be conveyed for 500yr flood
END DESCRIPTION:
XS GIS Cut Line= 6
     3193991.779    13974316.231     3192843.327    13974358.766
     3190503.887    13974752.218      3190300.42    13975154.866
     3189589.379    13975475.317 3187113.566549813976942.3963287
#Sta/Elev= 30
       0   80.38  208.14   79.35   437.3   68.61 1358.79   64.61 1496.35   68.88
  1896.1   65.51 2205.33   58.01 2598.36   61.74 2897.01   57.02  3096.9    62.2
 3477.32   60.97 3536.01   50.45 3616.73   55.96  3626.7      49  3642.7    46.6
  3656.7    38.4  3673.7    37.7  3796.7    46.2  3856.7    46.2 3941.45   59.09
 4110.46    56.2 4416.66    58.5 4538.02   54.53 4734.91   55.44 4899.33   70.07
 5025.36   67.19 5192.89   70.41 5971.65   66.96    7381      70    7641      74
#Mann= 3 ,-1 , 0
       0     .12       0  3642.7     .05       0  3796.7     .12       0
Bank Sta=3642.7,3796.7
XS Rating Curve= 0
Exp/Cntr=.3,.1

Type RM Length L Ch R = 1 ,94407.89,829.57,1525.75,1548.96
BEGIN DESCRIPTION:
411v20
Bank Station offset =      1632
ROB flow will be conveyed for 500yr flood
END DESCRIPTION:
XS GIS Cut Line= 6
     3191833.114    13971838.551      3189600.06    13974107.487
     3189591.644    13974404.846     3189387.336    13974677.781
     3187813.531    13976283.487 3187065.164138313976916.7234134
#Sta/Elev= 30
       0   80.01  672.96   80.82 1024.09   62.49  1347.2   55.74 1436.84   61.14
 1621.16   63.54 1790.08   61.35 2304.24   63.39 2459.89   60.45 2608.53   48.97
 2680.15   57.16  2741.5   60.07 2861.31   57.14 3047.53   60.05 3188.88   58.01
 3238.88   60.81 3267.88   48.71 3276.88   42.31 3367.88   39.61 3410.88   40.51
 3417.88   46.61 3440.88   48.41 3452.88   54.61 3513.81   57.94 3636.44   50.88
 3797.25   48.69 4010.01   65.54 4081.85   66.84 6264.76   66.23    7064      74
#Mann= 3 ,-1 , 0
       0     .12       0 3238.88     .05       0 3452.88     .12       0
Bank Sta=3238.88,3452.88
XS Rating Curve= 0
Exp/Cntr=.3,.1

Type RM Length L Ch R = 1 ,92882.15,1751.77,1538.72,830.92
BEGIN DESCRIPTION:
411v21
Bank Station offset =      2563
block on ROB to close cross section
END DESCRIPTION:
XS GIS Cut Line= 6
     3191301.423    13971625.875     3189680.506    13972865.869
     3189183.064    13972854.432     3188749.307    13973189.046
     3187845.433    13974348.132     3187494.517     13974730.95
#Sta/Elev= 30
       0   78.83  332.86   81.08  544.33   77.16  593.84    81.4  801.15   78.28
   891.2   81.66  997.78   80.71 1348.81    55.3 1450.67   59.79 2062.21   56.48
 2092.57    58.3 2122.57   68.54 2167.57   47.86 2233.23   50.81 2294.14    51.6
 2348.14    43.7 2357.14    39.5 2437.14    36.1 2448.14    44.3 2478.14    58.2
 2668.25   53.04 2815.53   57.25 2847.03   54.35 3019.53   54.44 3215.77   62.26
 3629.85   61.88 3861.86   70.01 4080.25   65.52 4354.76   70.05 5075.53   67.77
#Mann= 4 ,-1 , 0
       0     .12       0 2233.23     .05       0 2478.14     .12       0
 3861.86     .99       0
#Block Obstruct= 2 , 0
       0                 4354.76       0   70.05
Bank Sta=2294.14,2478.14
XS Rating Curve= 0
Exp/Cntr=.3,.1

Type RM Length L Ch R = 1 ,91343.42,977.67,1256.12,1651.13
BEGIN DESCRIPTION:
411v22
Bank Station offset =      3298
END DESCRIPTION:
XS GIS Cut Line= 6
     3189217.195    13970828.339     3188195.201    13972028.836
     3188397.901    13972224.297     3188419.659    13972338.341
     3186994.727    13974263.062 3185722.625574113976330.2258825
#Sta/Elev= 30
       0   75.33  453.93   71.58  571.85   66.84 1102.21   62.79 1237.22   55.94
 1412.38   55.24 1523.75   47.64 1563.13    51.2 1577.03   56.26 1602.03   53.96
 1666.03   42.36 1702.03   32.06 1740.03   38.46 1782.53   40.16 1795.03   46.86
 1812.03   50.96 1858.16   50.12 2006.19   48.55 2145.79   54.87 2220.99   45.31
 2259.37   44.49 2337.64   49.08 2733.26    60.8 3465.16   61.28 3642.42   67.65
  3809.3   68.53  4368.2   66.25 4613.08   68.36 4764.63   65.68    6800      68
#Mann= 4 ,-1 , 0
       0     .12       0 1602.03     .04       0 1858.16     .12       0
  3809.3     .99       0
Bank Sta=1602.03,1812.03
XS Rating Curve= 0
Exp/Cntr=.3,.1

Type RM Length L Ch R = 1 ,90087.30,1219.92,1493.05,1029.89
BEGIN DESCRIPTION:
411v23
Bank Station offset =      3127
block on ROB to close cross section
END DESCRIPTION:
XS GIS Cut Line= 6
     3188919.448    13970041.436      3188228.25    13970583.761
     3187387.646    13971334.193     3185357.119     13973337.92
     3184995.569    13973742.005     3184793.527    13973858.977
#Sta/Elev= 30
       0   77.81    89.4   77.13  186.33   70.85   248.2   76.03  704.54   77.16
 1106.51   63.18 1410.66   64.64 1506.21   59.67 1624.36   61.79 1757.17   55.79
  1771.8   53.73 1774.66    49.5 1814.66    53.2 1852.66      41 1872.66    37.7
 1933.66    39.1 1942.66    45.1 1958.66    49.2 2028.82   50.71  2181.7   58.77
  2202.5   55.84 2530.96   50.33 2751.26   56.53 3197.49   51.63 3288.33   54.84
 3452.07   52.88 3565.17   57.27 4559.16   55.27 4859.83   65.43  5635.6   66.11
#Mann= 3 ,-1 , 0
       0     .12       0 1814.66     .04       0 2028.82     .12       0
#Block Obstruct= 2 , 0
       0                 5296.06       0   67.79
Bank Sta=1814.66,1958.66
XS Rating Curve= 0
Exp/Cntr=.3,.1

Type RM Length L Ch R = 1 ,88594.25,923.1,1380.36,1545.86
BEGIN DESCRIPTION:
411v24
Bank Station offset =      2660
END DESCRIPTION:
XS GIS Cut Line= 6
     3188525.997     13969605.45     3187834.799    13969807.492
     3186941.558    13970158.408     3186295.583     13970743.83
     3185144.443    13972327.707     3184229.935    13973901.512
#Sta/Elev= 30
       0   75.46  235.11   74.92  469.85   68.01  720.12   69.81 1066.49   62.15
 1387.34   62.39 1602.69   70.29 1917.89   61.25  2108.4   62.61 2235.47   58.09
 2260.47   47.89 2275.47   36.89 2290.47   31.59 2340.47   31.19 2370.47   33.19
 2380.47   41.39 2400.47   48.49 2435.47   44.69 2470.47   48.89 2642.78   52.03
 2679.88    48.2 2824.44   46.24 2871.65   51.34 3272.62   52.29 3459.64   48.12
 3821.45   56.47 4788.31   54.23    5164   64.43 6009.96   64.61 6332.79   68.65
#Mann= 4 ,-1 , 0
       0     .99       0 1602.69     .12       0 2260.47     .04       0
 2470.47     .12       0
Bank Sta=2260.47,2400.47
XS Rating Curve= 0
Exp/Cntr=.3,.1

Type RM Length L Ch R = 1 ,87213.89,837.62,1915.68,1942.11
BEGIN DESCRIPTION:
411v25
Bank Station offset =      2281
END DESCRIPTION:
XS GIS Cut Line= 6
     3187739.094    13969499.112     3186856.488    13969637.351
     3185973.881    13969860.661     3185312.815    13970343.765
     3183762.047    13971157.987     3182975.144    13971721.579
#Sta/Elev= 30
       0   67.39  268.47   73.12  540.65   61.58 1428.34   62.19 1625.45   52.19
 1778.97   49.53 1846.33   52.44 2050.24   51.82 2084.24   46.26 2135.99    50.8
 2427.31   52.18 2634.15   49.18 2649.15   39.38 2679.15   37.68 2719.15   30.88
 2759.15   34.08 2774.15   41.28 2779.15   50.58 2845.37   50.42 2882.55   45.81
 2938.36   53.06 3216.24    56.4 3455.05   53.37 3890.95   53.21 4049.07   61.85
 4286.57   61.85 4425.04   57.49 4676.61    65.4 5075.58   62.59 5343.09   65.21
#Mann= 5 ,-1 , 0
       0     .12       0 2634.15     .04       0 2779.15     .12       0
 4286.57     .99       0 4676.61     .12       0
#Block Obstruct= 2 , 0
       0                    4700       0      66
Bank Sta=2634.15,2779.15
XS Rating Curve= 0
Exp/Cntr=.3,.1

Type RM Length L Ch R = 1 ,85298.22,1479.93,1351.48,850.3
BEGIN DESCRIPTION:
411v26
Bank Station offset =      2313
END DESCRIPTION:
XS GIS Cut Line= 6
     3187951.771    13969116.294     3185761.204     13969020.59
     3185180.316    13968884.081     3184580.851    13968839.815
     3181497.043    13969435.309     3181231.198    13969616.084
#Sta/Elev= 30
       0   69.74  184.74      64 1024.88   61.73 1054.47   56.77 1089.93   60.64
 1327.34   65.16  1680.5   61.35 1854.05   52.83  2547.3   49.84  2557.3   45.74
  2572.3   48.54  2622.3   34.64  2687.3   29.44  2712.3   36.74  2727.3   50.74
  2792.3   49.64 2990.86   49.87 3139.55   53.35 3546.72   52.47 3721.52   56.82
 4015.73   58.81 4240.03   52.41 4419.14   56.84 4876.99   55.58 5059.77   58.42
 5294.55   55.73 5467.45   61.06 5989.63   61.11 6302.25   68.66 6859.47   69.46
#Mann= 5 ,-1 , 0
       0     .12       0 1024.88     .99       0 1089.93     .12       0
  2547.3     .04       0  2792.3     .12       0
Bank Sta=2572.3,2727.3
XS Rating Curve= 0
Exp/Cntr=.3,.1

Type RM Length L Ch R = 1 ,83946.74,916.6,1363.39,1037.34
BEGIN DESCRIPTION:
411v27
Bank Station offset =      3614
END DESCRIPTION:
XS GIS Cut Line= 6
     3187228.671    13967680.729     3186144.022    13967670.095
     3185727.837    13967847.109     3185165.711    13967957.208
     3182645.496    13968382.561     3181284.367    13968552.702
#Sta/Elev= 30
       0   76.68  292.26   75.98  523.75   69.34  773.18   54.09  994.34   50.94
 1207.56   51.09 1264.74   46.73  1329.4   47.91 1340.74   47.63 1341.48   49.41
 1351.48   35.91 1361.48   29.11 1386.48   26.91 1501.48   45.51 1536.48   46.51
 1618.24   43.45 1677.99   46.54 2454.05   46.61 2500.08   53.66 2555.98   56.79
 2786.49   59.84 3438.92   56.38 3514.98   58.33 3603.85   55.46 3805.47   54.89
 4070.52   58.71 4514.67   55.74 5273.54   62.58 5718.63   62.21 6042.71   68.74
#Mann= 3 ,-1 , 0
       0     .12       0  1329.4     .04       0 1510.68     .12       0
Bank Sta=1341.48,1501.48
XS Rating Curve= 0
Exp/Cntr=.3,.1
